--- StnclCrk.prj (project) ---

Proj Title=StnclCrk
Current Plan=p01
Default Exp/Contr=0,0
English Units
Geom File=g01
Flow File=f01
Plan File=p01
BEGIN DESCRIPTION:
END DESCRIPTION:
DSS Export Rating Curves= 0
DSS Export Rating Curve Sorted= 0
DSS Export Volume Flow Curves= 0
DXF OffsetX= 0
DXF OffsetY= 0
DXF ScaleX= 0
DXF ScaleY= 0

--- StnclCrk.p01 (plan) ---

Plan Title=Floodplain
Program Version=4.00
Geom File=g01
Flow File=f01
K Sum by GR=0
Std Step Tol=0.01
Critical Tol=0.01
Num of Std Step Trials=20
Max Error Tol=0.3
Flow Tol Ratio=0.001
Split Flow NTrial=30
Split Flow Tol=0.02
Split Flow Ratio=0.02
Log Output Level=0
Friction Slope Method=1
Unsteady Friction Slope Method=2
Unsteady Bridges Friction Slope Method=1
Global Log Level=0
CheckData=False
Run HTab=0
Run UNet=0
Run PostProcess=0
UNET Theta=0
UNET Theta Warmup=0
UNET ZTol=0
UNET ZSATol=0
UNET MxIter=0
UNET MaxInSteps=0
UNET DtIC=0
UNET DtMin=0
UNET MaxCRTS=0
UNET WFStab=0
UNET SFStab=0
UNET WFX=0
UNET SFX=0
UNET DSS MLevel=0
UNET DZMax Abort=0
UNET Convert EG Bridges=0
UNET Use Existing IB Tables=0
UNET Froude Limit=0
UNET Froude Power=0
Write IC File=0
Echo Input=False
Echo Output=False
Write Detailed=0

--- StnclCrk.f01 (steady flow) ---

Flow Title=NFF Regression Equation
Program Version=4.00
Number of Profiles=1
Profile Names=P100yr
River Rch & RM=StnclCrk,Main      ,43219.1
861.5325
River Rch & RM=StnclCrk,Main      ,41804.7
897.6510
River Rch & RM=StnclCrk,Main      ,41481.5
1016.146
River Rch & RM=StnclCrk,Main      ,41316.2
1018.951
River Rch & RM=StnclCrk,Main      ,40611.1
1273.303
River Rch & RM=StnclCrk,Main      ,39019.1
1303.333
River Rch & RM=StnclCrk,Main      ,37519.1
1444.058
River Rch & RM=StnclCrk,Main      ,36643.8
1544.226
River Rch & RM=StnclCrk,Main      ,32772
1692.160
River Rch & RM=StnclCrk,Main      ,29952.3
1787.382
River Rch & RM=StnclCrk,Main      ,29457.2
2369.650
River Rch & RM=StnclCrk,Main      ,25794.5
2443.640
River Rch & RM=StnclCrk,Main      ,16550.5
2701.575
River Rch & RM=StnclCrk,Main      ,16226.2
3041.287
River Rch & RM=StnclCrk,Main      ,11002.9
3121.711
River Rch & RM=StnclCrk,Main      ,10692
3629.115
River Rch & RM=StnclCrk,Main      ,248.3
3881.209
Boundary for River Rch & Prof#=StnclCrk,Main      ,1
Up Type=0
Dn Type=3
Dn Slope=0.001151

--- StnclCrk.g01 (geometry) ---

Geom Title=USGS 3m DEM
Program Version=4.10

River Reach=StnclCrk        ,Main
Reach XY= 30
     1904974.588      236935.924     1905550.108      234947.643
     1903325.302      232890.276     1902207.714      233178.175
     1900543.937      231805.947     1899747.126      231511.405
     1899111.453      230687.776     1899474.809      228838.129
       1897294.3      228193.431     1896743.298      227630.743
     1895955.255      227828.759      1894944.74      227450.696
     1894061.322      227565.706     1893460.817      226874.067
     1890738.305      227039.404     1890005.142      227406.938
     1889540.152      228038.696     1888035.713      228512.883
     1887078.326      228350.099     1886463.499       227860.36
     1882759.087      229501.727     1881832.943       228842.67
     1881685.693      227331.709     1881067.833      226851.247
     1880921.032      225881.992     1880049.564      224522.156
     1878948.879      223998.574     1879088.233      223525.739
     1880090.164      222911.141     1880284.007      221527.444

Type RM Length L Ch R = 1 ,43219.1 ,252.2,254,256
XS GIS Cut Line= 3
     1905519.707      236967.291     1904975.231      236925.944
     1904430.372       236890.79
#Sta/Elev= 30
       0 2280.76    89.4  2262.2   129.1 2248.16   158.8 2241.91   208.5  2217.9
   218.4 2208.54   287.9 2166.58   297.8 2155.45   367.3 2114.09   377.3 2103.69
   387.2  2096.6   446.8 2059.06   456.7 2045.51   466.6 2034.74   496.4 2010.43
   506.3 2004.58   516.3 2001.77   538.5 1999.59     546 1999.02   553.5  1999.3
     695 2008.01   714.8 2015.33   774.4 2028.33   794.2 2041.96   814.1 2052.17
   933.2 2100.89   953.1 2113.86  1022.6 2146.46  1032.5 2154.43    1092 2183.04
#Mann= 3 , 0 , 0
       0      .1       0   538.5    .045       0   553.5      .1       0
Bank Sta=538.5,553.5
XS Rating Curve= 0 ,0
Exp/Cntr=0.3,0.1

Type RM Length L Ch R = 1 ,42965   ,342.9,345.9,348.9
XS GIS Cut Line= 2
     1905525.851       236756.33     1904425.316      236586.189
#Sta/Elev= 30
       0 2221.22    49.7 2203.48    69.6 2190.89   129.3 2167.35   149.1 2155.04
   208.8 2134.99   228.7  2123.4   298.3 2095.95   308.2 2088.54   377.8 2060.57
   387.8 2052.43   467.3 2016.84   477.3 2009.22   487.2 2004.79   540.4 1994.55
   555.4 1993.35   556.8 1993.32   686.1 2000.21     706  2003.5   765.6 2022.58
   795.4 2037.62   805.4 2047.08     875 2083.38   884.9 2093.86   964.5 2137.44
   974.4 2147.33  1004.2 2164.96  1024.1 2174.73    1044 2177.21  1113.6 2222.79
#Mann= 3 , 0 , 0
       0      .1       0   540.4    .045       0   555.4      .1       0
Bank Sta=540.4,555.4
XS Rating Curve= 0 ,0
Exp/Cntr=0.3,0.1

Type RM Length L Ch R = 1 ,42619.1 ,171.4,172.8,174.3
XS GIS Cut Line= 3
     1905592.593      236493.379      1905069.09      236338.211
     1904544.576      236186.559
#Sta/Elev= 30
       0 2306.68    39.7 2282.41    59.6 2264.64   119.1 2229.97   129.1  2221.8
     139 2211.14   218.4 2159.34   228.3 2148.42   238.3 2141.04   297.8 2105.42
   317.7 2088.92   387.2 2052.67   397.1 2043.32   456.7 2014.25   476.5 2006.74
   506.3 2002.95   516.2 1999.95   538.5  1989.1   553.5 1986.99   555.9 1986.98
   575.8 1989.68   625.4 1991.21   645.3 1993.73     814 2031.83   893.5 2054.05
   913.3 2062.17   972.9 2079.39  1012.6  2095.4  1072.2 2123.42    1092 2137.21
#Mann= 3 , 0 , 0
       0     .06       0   538.5    .045       0   553.5     .06       0
Bank Sta=538.5,553.5
XS Rating Curve= 0 ,0
Exp/Cntr=0.3,0.1

Type RM Length L Ch R = 1 ,42446.4 ,123.1,125.2,126.3
XS GIS Cut Line= 3
     1905527.354      236372.606     1905176.016      236194.409
     1904714.727      236026.323
#Sta/Elev= 30
       0 2231.96    68.9 2190.24    88.6  2172.8   157.6 2130.74   177.3 2112.86
     197 2100.69   246.2 2073.34   256.1 2066.02   265.9 2056.28   285.6 2044.76
   344.7 2011.62   354.6 2007.79   384.1 2004.45   393.9 2001.57   423.4  1986.6
   429.2 1985.05     443  1983.6   444.2 1983.72   521.6 1987.88   541.2 1990.07
     610 2004.07   629.6 2010.19   668.9 2018.72   698.3 2031.33   708.2  2038.5
   727.8  2045.9   776.9 2067.81   796.5 2080.33   875.1  2114.7   884.9 2120.71
#Mann= 3 , 0 , 0
       0     .06       0   429.2    .045       0   444.2     .06       0
Bank Sta=429.2,444.2
XS Rating Curve= 0 ,0
Exp/Cntr=0.3,0.1

Type RM Length L Ch R = 1 ,42321   ,266.6,266.2,266.8
XS GIS Cut Line= 3
     1905644.288       236392.94     1905218.985      236080.667
     1904721.046      235868.347
#Sta/Elev= 30
       0 2298.66    19.9 2281.93    39.8 2278.25   119.5 2231.23   129.4 2224.66
   139.4 2215.16   189.2 2189.63     219 2172.18     229 2165.19   238.9    2155
   318.6  2103.3   328.5 2094.99   338.5 2083.54   358.4 2073.88   418.1  2034.3
     438 2017.13   507.7 2000.59     539 1983.47     554 1981.34     626  1980.6
   704.8 1983.63   724.5 1991.03   793.4 2009.31   891.8  2053.9   911.5 2066.92
   980.4 2097.31    1000 2112.45  1029.6 2127.88  1039.4 2132.24    1069 2136.62
#Mann= 3 , 0 , 0
       0     .06       0     539    .045       0     554     .06       0
Bank Sta=539,554
XS Rating Curve= 0 ,0
Exp/Cntr=0.3,0.1

Type RM Length L Ch R = 1 ,42055.2 ,250.4,250.1,249.8
XS GIS Cut Line= 2
     1905845.628      236082.234     1904836.379      235627.653
#Sta/Elev= 30
       0  2171.9    29.9 2173.02   119.7 2160.48   169.5 2151.38   199.4 2151.99
   229.4 2146.06   249.3 2136.52   259.3 2133.52   329.1 2100.39     349 2088.67
   378.9 2075.24   428.8  2042.3   448.7 2026.28   508.6 1995.07   518.6 1988.54
   528.5 1978.34   538.5 1975.85   546.8 1975.88   561.8 1975.68   608.3 1975.24
   658.2 1976.06   757.9 1986.48   787.8 1993.84   807.7 2001.95   867.6 2007.35
   897.5  2017.2   967.3 2030.27   987.2 2036.64    1057 2053.36  1106.9 2077.76
#Mann= 3 , 0 , 0
       0      .1       0   546.8    .045       0   561.8      .1       0
Bank Sta=546.8,561.8
XS Rating Curve= 0 ,0
Exp/Cntr=0.3,0.1

Type RM Length L Ch R = 1 ,41804.7 ,335.3,323.2,311.6
XS GIS Cut Line= 2
     1905972.366      235866.679     1904946.162      235423.074
#Sta/Elev= 30
       0  2032.5    89.8  2024.8   119.8 2027.61   189.7 2018.93   209.6 2017.96
   289.5 2009.88   309.4 2009.62   339.4 2006.96   369.3 2008.35   389.3  2005.6
   449.2 2002.34   469.2 1998.59   479.1 1994.74   489.1 1988.82   533.2 1972.65
   548.2 1971.27   658.8 1972.64   718.7 1970.59   748.6 1974.69   818.5  2001.4
   838.5 2006.84   848.5 2011.32   858.4 2013.33   888.4 2015.12   908.4 2017.65
   928.3 2021.72  1008.2 2041.89  1028.1 2050.77    1108 2072.82    1118 2077.34
#Mann= 3 , 0 , 0
       0      .1       0   533.2    .045       0   548.2      .1       0
Bank Sta=533.2,548.2
XS Rating Curve= 0 ,0
Exp/Cntr=0.3,0.1

Type RM Length L Ch R = 1 ,41481.5 ,164.2,165.2,165.7
XS GIS Cut Line= 3
     1906072.024      235292.018      1905525.47      235355.952
     1904960.884      235401.282
#Sta/Elev= 30
       0 2187.57      60 2175.24   130.1 2170.28   160.1 2160.06   210.1 2136.99
   220.1 2128.44   230.1 2123.42   290.2 2097.63   300.2 2089.79   310.2 2084.52
   370.2 2057.13   390.2 2042.74   450.2 2012.99   470.2 2007.63   490.2 1991.64
   534.9 1968.93   549.9 1966.88   659.6 1966.26   689.4 1968.11   729.2 1975.73
   768.9 1974.36   788.8 1975.75   828.5 1997.81   848.4 2005.78   927.9 2015.45
   957.7 2023.93   967.6 2028.72  1037.2 2047.51  1047.1 2052.42  1116.7 2071.46
#Mann= 3 , 0 , 0
       0      .1       0   534.9    .045       0   549.9      .1       0
Bank Sta=534.9,549.9
XS Rating Curve= 0 ,0
Exp/Cntr=0.3,0.1

Type RM Length L Ch R = 1 ,41316.2 ,501.8,482.8,453.5
XS GIS Cut Line= 3
     1906139.035      234909.119     1905656.382      235182.178
     1904978.186      235243.018
#Sta/Elev= 30
       0 2024.13    49.5  2028.6    69.3  2027.8   118.8 2032.55   158.4 2026.09
   227.8  2036.4   247.6 2036.15     307 2043.17   326.8 2039.34   336.7 2039.53
   386.2 2045.33   415.9 2046.36   475.3 2040.59   554.5 2027.58   584.2 2010.63
   603.9 2004.63   623.6 1985.85   633.5 1981.36   643.4 1979.15   682.8 1977.39
   720.7 1965.38   732.2 1964.54   735.7 1964.61   811.1 1965.14   899.9 1972.41
   929.5 1972.48  1008.5  1993.8  1038.1  2004.3  1176.2 2036.08  1235.5 2055.49
#Mann= 3 , 0 , 0
       0      .1       0   720.7    .045       0   735.7      .1       0
Bank Sta=720.7,735.7
XS Rating Curve= 0 ,0
Exp/Cntr=0.3,0.1

Type RM Length L Ch R = 1 ,40833.3 ,221.4,222.1,222.9
XS GIS Cut Line= 4
     1906050.569      234761.254      1905426.95        234843.1
     1905234.249      235068.005     1904978.186      235243.018
#Sta/Elev= 30
       0 2001.23    49.9 2011.87   119.8  2015.7   149.8 2019.73   199.7  2028.6
   219.6  2034.4   289.5 2039.08   359.4 2034.63   419.3 2036.24   439.3 2034.37
   479.2 2026.63   539.1 2022.82   559.1 2018.48     619 2002.02     629    1998
   658.6    1978   678.3 1970.28   688.2 1962.83   696.5 1960.45   707.9 1959.51
   711.5 1959.69   846.2 1968.47   925.1  1969.8   965.2 1973.15   975.2 1975.69
  1005.2 1994.83  1035.2    2008  1155.2 2030.96  1185.3 2041.66  1235.3 2055.49
#Mann= 3 , 0 , 0
       0      .1       0   696.5    .045       0   711.5      .1       0
Bank Sta=696.5,711.5
XS Rating Curve= 0 ,0
Exp/Cntr=0.3,0.1

Type RM Length L Ch R = 1 ,40611.1 ,259.6,257.1,254.7
XS GIS Cut Line= 2
     1905341.574      234618.444      1904839.69      235148.967
#Sta/Elev= 30
       0 2063.93      10 2055.54      20  2052.9      40 2050.86      50 2045.97
      80 2026.46     100 2018.43     120  2001.3   150.1 1981.54   172.9  1964.4
   180.1 1959.96   187.9 1959.05   190.1 1958.79   230.1 1967.14   250.1 1969.68
   290.1 1965.57   360.2 1965.54   370.2 1969.17   410.2 1994.49   440.2 2011.24
   460.2 2016.21   520.2 2025.18   560.2 2040.24   580.2 2050.93   590.2  2053.2
   650.3 2074.16   680.3 2078.23   690.3 2080.81   710.3 2089.89   730.3 2096.77
#Mann= 3 , 0 , 0
       0      .1       0   172.9    .045       0   187.9      .1       0
#XS Ineff= 2 , 0
                          251.36         1969.45
Permanent Ineff=
       F       F
Bank Sta=172.9,187.9
XS Rating Curve= 0 ,0
Exp/Cntr=0.3,0.1

Type RM Length L Ch R = 1 ,40354   ,114.6,119.4,124.2
XS GIS Cut Line= 3
     1905317.987      234190.696     1904978.953      234654.083
     1904688.503      235110.537
#Sta/Elev= 30
       0 2153.35    89.1 2127.65   118.8 2115.46   158.4 2106.92   227.7 2085.45
   257.4  2072.1   287.1  2065.9   346.5 2041.92   366.3 2038.04     396 2024.31
   475.2  1976.8     495 1971.43   514.8 1959.14   519.8 1958.22   524.7 1957.32
   534.8 1958.71   574.2 1968.54   662.7 1963.41     702 1989.33   711.9 1991.79
   741.4 2012.69   751.2 2016.78   790.6 2027.63   820.1 2042.16   829.9 2043.15
   869.3 2062.48   938.1 2076.02  1026.7 2105.76  1046.3 2109.22  1115.2 2145.85
#Mann= 3 , 0 , 0
       0      .1       0   519.8    .045       0   534.8      .1       0
#XS Ineff= 2 , 0
                          584.64         1969.17
Permanent Ineff=
       F       F
Bank Sta=519.8,534.8
XS Rating Curve= 0 ,0
Exp/Cntr=0.3,0.1

Type RM Length L Ch R = 1 ,40234.1 ,111.4,118.3,125.2
XS GIS Cut Line= 2
     1905022.094      234462.948     1904570.392      234853.308
#Sta/Elev= 30
       0 2023.63    19.9 2011.93    39.8 2003.03    49.8 2001.28    59.7 1998.53
    99.5 1980.73   109.4 1975.94   119.4 1969.96   139.3 1960.76   149.2 1956.79
     158 1955.68   159.2 1955.53     173 1958.27   179.1 1960.22     199 1962.61
   228.8 1960.96   258.7 1961.42   268.6 1964.02   278.6 1969.03   308.4 1986.18
   358.2 2012.89   368.2 2015.56   417.9 2020.96   427.8 2022.83   437.8 2025.74
   467.6 2031.67   537.3 2051.96   557.2 2054.29   567.2 2057.28     597 2068.78
#Mann= 3 , 0 , 0
       0     .06       0     158    .045       0     173     .06       0
#XS Ineff= 2 , 0
                          199.22         1962.76
Permanent Ineff=
       F       F
Bank Sta=158,173
XS Rating Curve= 0 ,0
Exp/Cntr=0.3,0.1

Type RM Length L Ch R = 1 ,40115.8 ,457.8,451.9,445.9
XS GIS Cut Line= 2
     1905121.672      234357.468     1904548.747      234600.119
#Sta/Elev= 30
       0 2078.16    29.6 2069.52    39.5 2068.14    88.9 2064.25    98.8 2062.33
   108.6 2058.46   118.5 2052.35   128.4 2042.91   138.3 2036.63   167.9  2022.9
   207.4 2006.04   217.3 1998.54   286.4 1968.56   296.3 1963.68   306.2 1956.55
     316 1953.24   321.5 1952.71   325.9 1952.28   336.5 1953.07   365.4 1959.23
     395 1960.94   414.8 1960.21   424.7 1960.72   434.6 1963.08   464.2 1974.79
   483.9 1985.28   543.2 2008.83   553.1 2011.44   562.9 2016.17   622.2 2038.74
#Mann= 3 , 0 , 0
       0     .06       0   321.5    .045       0   336.5     .06       0
Bank Sta=321.5,336.5
XS Rating Curve= 0 ,0
Exp/Cntr=0.3,0.1

Type RM Length L Ch R = 1 ,39663.9 ,345.1,344.8,344.5
XS GIS Cut Line= 2
     1904919.404      233850.919      1904064.46      234532.927
#Sta/Elev= 30
       0 2235.57     9.9 2226.39    99.4 2176.31   109.4 2166.92   198.8 2121.04
   218.7 2105.87   298.3 2066.36   318.2 2051.69   397.7 2009.96   407.6  2006.8
   447.4 1983.18     507 1956.26   526.9  1943.7   531.8 1943.22   536.9 1942.72
   546.8 1943.75   586.6 1950.51   636.3 1950.75   656.2 1956.28   705.9 1990.85
   765.6 2019.03   825.2 2052.34   835.2 2056.26     865  2057.7   884.9 2064.88
   914.7 2079.72   984.3 2123.18   994.2 2127.98  1014.1 2133.24  1093.6 2176.87
#Mann= 3 , 0 , 0
       0     .06       0   531.8    .045       0   546.8     .06       0
Bank Sta=531.8,546.8
XS Rating Curve= 0 ,0
Exp/Cntr=0.3,0.1

Type RM Length L Ch R = 1 ,39319.1 ,298.9,300,298.1
XS GIS Cut Line= 3
     1904704.134      233572.871     1904281.941      233919.091
     1903859.747      234265.311
#Sta/Elev= 30
       0 2226.81    39.7 2210.56    59.6 2196.02    99.3 2171.73   119.1 2164.96
   148.9  2145.1   158.8  2136.1   228.3 2089.98   347.4 2028.98   367.3 2014.91
   456.6 1977.87   476.5 1965.89   538.5 1938.55   553.5 1936.67   555.9 1936.56
   595.6 1946.34   635.4 1946.11   645.3 1947.82   655.2 1953.74   665.1 1963.68
     675 1977.48   704.8 1995.45   734.6 2008.58     814 2049.11   873.6  2058.7
     953 2104.45   972.9 2110.01   992.7 2123.45  1072.2 2167.61    1092  2181.5
#Mann= 3 , 0 , 0
       0     .06       0   538.5    .045       0   553.5     .06       0
Bank Sta=538.5,553.5
XS Rating Curve= 0 ,0
Exp/Cntr=0.3,0.1

Type RM Length L Ch R = 1 ,39019.1 ,304.7,300.1,301.4
XS GIS Cut Line= 3
     1904543.081      233354.389     1904104.003      233678.563
     1903710.465      234061.011
#Sta/Elev= 30
       0 2189.97    19.8 2185.79    39.7 2177.37   158.8 2101.12   178.6 2092.39
   198.5 2078.89   238.2 2058.19   327.5 2031.31   367.2 2005.42   446.6 1969.66
   466.4 1958.03   538.3 1931.23   545.8 1930.68   553.3 1932.07   625.6 1940.55
   635.6 1943.78   665.5 1962.29   725.4 2006.33   745.3 2015.13   765.3 2028.23
   795.2 2053.22   805.2 2058.86   825.2 2062.22   835.1 2067.25   855.1 2081.39
     885 2095.54     905 2110.96   994.8 2157.81  1014.7 2173.97  1094.5 2221.69
#Mann= 3 , 0 , 0
       0     .06       0   538.3    .045       0   553.3     .06       0
Bank Sta=538.3,553.3
XS Rating Curve= 0 ,0
Exp/Cntr=0.3,0.1

Type RM Length L Ch R = 1 ,38719.1 ,300.9,299.8,295.3
XS GIS Cut Line= 3
     1904285.135      233042.355      1903922.13      233448.945
     1903505.531      233810.078
#Sta/Elev= 30
       0 2241.03    29.7 2223.06    49.6 2216.29    69.4 2201.47     109 2178.29
   148.6 2146.96   168.5 2137.22   188.3 2117.91   237.8 2086.01   277.5 2063.18
     337 2034.12   426.1 1983.93   515.3  1928.8   525.2 1926.42   537.6 1926.66
   552.6  1928.6   594.3 1930.86   653.4 1938.73   682.9 1950.88   712.4 1970.36
     742 1981.22   761.6 1992.06   791.2 2003.34   820.7 2021.64   889.6 2052.83
   909.3 2055.71   988.1 2093.68  1007.8 2103.88  1027.5 2120.49  1096.4 2156.82
#Mann= 3 , 0 , 0
       0      .1       0   537.6    .045       0   552.6      .1       0
Bank Sta=537.6,552.6
XS Rating Curve= 0 ,0
Exp/Cntr=0.3,0.1

Type RM Length L Ch R = 1 ,38419.1 ,159.9,158.5,157.7
XS GIS Cut Line= 3
     1904054.138      232819.409     1903705.939      233241.835
     1903370.717      233673.371
#Sta/Elev= 30
       0 2227.58    89.6 2192.19   119.4 2175.58   189.1 2128.62     209 2120.48
   228.9 2102.53   308.6  2047.9   328.5 2039.82   358.3 2016.78   398.1 1992.39
   517.6 1924.03   539.9 1924.89   554.9 1925.17     607 1925.11   646.8 1935.54
   686.5 1965.28   696.5 1971.33   706.4  1973.4     776 2019.73   805.8 2043.43
   845.5 2051.43   855.4 2056.52   895.2 2085.91     915 2104.76     925 2111.04
   934.9 2113.41  1024.3 2175.66  1044.2 2191.95  1064.1 2200.23  1093.9  2219.9
#Mann= 3 , 0 , 0
       0      .1       0   539.9    .045       0   554.9      .1       0
Bank Sta=539.9,554.9
XS Rating Curve= 0 ,0
Exp/Cntr=0.3,0.1

Type RM Length L Ch R = 1 ,38260.6 ,162.6,161.3,159.9
XS GIS Cut Line= 3
     1903923.585      232675.765      1903709.58      232972.338
     1903263.187      233585.433
#Sta/Elev= 30
       0 2145.67    29.6 2132.88    69.2 2128.15   118.6 2129.59   158.2 2126.04
   187.8 2127.26   247.1 2093.96   276.8 2081.73   296.5 2066.92   385.7 2014.92
   495.4 1946.97   525.4 1925.39   535.4 1922.05   551.4 1922.47   566.4 1923.08
   645.1 1921.39     685 1930.63     715 1949.88   734.9 1957.17   774.8 1988.08
   824.8 2022.53   844.7 2029.94   864.7 2041.58   884.6 2044.78   954.5 2089.99
   964.4 2090.53   974.4  2095.6  1064.2 2150.89  1084.2 2156.09  1124.1 2180.79
#Mann= 3 , 0 , 0
       0     .06       0   551.4    .045       0   566.4     .06       0
Bank Sta=551.4,566.4
XS Rating Curve= 0 ,0
Exp/Cntr=0.3,0.1

Type RM Length L Ch R = 1 ,38099.3 ,292.7,288.8,280.5
XS GIS Cut Line= 2
     1903572.185      232873.624     1903318.451      233272.349
#Sta/Elev= 30
       0 2007.39     9.8 2003.58    19.7 2000.49    39.4 1989.18    59.1 1973.67
    88.6 1955.96   108.3 1943.83   118.2 1940.72     128 1937.25   137.8 1930.74
   147.7 1923.55   157.5    1920   158.8 1919.94   167.4 1919.56   173.8 1919.84
   216.6 1921.85   246.2 1921.25   295.4 1918.71   305.2 1918.55   315.1 1919.55
   324.9 1922.22   334.8 1925.95   344.6 1927.82   354.5  1931.6   374.2 1944.97
   393.8 1956.85   423.4 1977.54   452.9 1997.87   462.8 2000.66   472.6 2004.53
#Mann= 3 , 0 , 0
       0     .06       0   158.8    .045       0   173.8     .06       0
Bank Sta=158.8,173.8
XS Rating Curve= 0 ,0
Exp/Cntr=0.3,0.1

Type RM Length L Ch R = 1 ,37810.5 ,303.5,291.4,286.4
XS GIS Cut Line= 4
     1903382.676       232451.65     1903255.754       232772.05
     1903276.517      233115.569     1903197.512      233559.405
#Sta/Elev= 30
       0 2005.33   137.8 1978.17   157.5 1977.35   226.5 1961.06   265.8 1957.24
   324.9  1942.1   364.3 1936.68   393.8 1928.94   462.6 1921.54   482.3 1915.52
     502 1913.95   507.4 1913.97   522.4 1914.31   659.3 1914.97   688.8 1921.98
     728 1946.79   747.6 1953.45   816.2 2001.17   835.8 2007.85   865.2 2028.44
   894.6 2035.24     924 2051.73   933.8 2052.58   943.6 2057.52  1012.2 2098.21
  1031.8 2104.49  1110.2 2155.67    1120 2161.18  1129.8 2162.13  1139.6 2168.73
#Mann= 3 , 0 , 0
       0      .1       0   507.4    .045       0   522.4      .1       0
Bank Sta=507.4,522.4
XS Rating Curve= 0 ,0
Exp/Cntr=0.3,0.1

Type RM Length L Ch R = 1 ,37519.1 ,189.8,188.4,184.1
XS GIS Cut Line= 3
      1902980.99       232432.61      1903013.04      233044.803
     1902964.649      233576.698
#Sta/Elev= 30
       0 2152.85    49.4 2117.87    69.2 2109.22   108.8 2072.64   128.5 2059.58
   148.3 2048.44   168.1 2043.52   247.2 2001.07   257.1  2000.1   346.1 1943.84
     356 1943.39   375.7 1930.97   454.8 1923.36     524 1910.88   603.1 1907.17
   605.5  1907.5   620.5 1911.21   652.6 1920.38   711.9 1957.72   731.7 1963.87
     801 2007.56   840.5 2016.57   860.3  2039.1   899.9 2057.81   919.6 2061.59
   939.4 2070.58  1008.6 2112.24  1018.5 2112.02  1097.7 2149.93  1147.1 2156.06
#Mann= 3 , 0 , 0
       0      .1       0   605.5    .045       0   620.5      .1       0
Bank Sta=605.5,620.5
XS Rating Curve= 0 ,0
Exp/Cntr=0.3,0.1

Type RM Length L Ch R = 1 ,37330.7 ,327,324.6,239.1
XS GIS Cut Line= 3
     1902874.061      232411.452     1902826.602       232913.36
     1902859.722      233560.647
#Sta/Elev= 30
       0 2141.83    79.1 2090.32      89 2089.24   118.6 2078.98   138.4 2066.94
     168 2045.17   177.9 2044.56   207.6 2028.38   247.1 2013.22   266.9 2006.99
   276.8 2006.83   286.7 2002.81   355.9 1959.17   365.8 1957.84   395.4 1940.14
   415.2 1930.61   454.7 1916.01   494.3 1910.72   584.3 1903.67   593.9 1903.49
   599.3 1903.91   693.6 1917.94   733.5 1938.54   753.4 1943.72   833.2    1987
   853.1 1993.44     913 2030.38   942.9  2038.3  1022.6 2070.24  1152.3 2083.94
#Mann= 3 , 0 , 0
       0      .1       0   584.3    .045       0   599.3      .1       0
Bank Sta=584.3,599.3
XS Rating Curve= 0 ,0
Exp/Cntr=0.3,0.1

Type RM Length L Ch R = 1 ,37006.1 ,354.3,361.7,369.2
XS GIS Cut Line= 3
     1902506.603      232471.135     1902658.095      233120.624
     1902795.466      233563.908
#Sta/Elev= 30
       0 2080.96      10 2075.38    19.9 2072.33    49.8 2050.88    69.7 2040.61
   109.5 2024.44   119.4 2023.84   149.3 2010.27   199.1 1990.94   248.8 1980.15
   348.4  1965.3   408.1  1963.6   418.1 1961.72   497.7 1911.41   527.6 1904.32
   572.8 1897.28   577.3 1897.03   587.8 1898.04   706.4 1917.24     736 1927.09
   785.4 1951.31   805.2 1956.76   834.8 1968.01   864.4 1975.57   923.6  1984.9
   943.4 1991.39     973 2006.46   982.9 2009.63  1061.9 2025.33    1131 2044.43
#Mann= 3 , 0 , 0
       0      .1       0   572.8    .045       0   587.8      .1       0
Bank Sta=572.8,587.8
XS Rating Curve= 0 ,0
Exp/Cntr=0.3,0.1

Type RM Length L Ch R = 1 ,36643.8 ,307.9,323.8,339.7
XS GIS Cut Line= 3
     1902358.776      232496.079     1902299.174      233226.784
     1902458.131      233661.937
#Sta/Elev= 30
       0 2101.59    49.5 2069.08    69.4 2063.28    79.3 2062.67    99.1 2057.83
   168.4 2031.68   188.2 2027.62   237.8 2004.72   257.6  1992.8   277.4 1987.75
   307.1 1975.73   376.5 1965.92   455.7 1940.53   465.6 1939.64   544.9  1905.5
   659.7 1894.31   673.7 1893.56   674.7 1893.74   683.6  1895.3   733.1 1912.27
   752.8 1915.83   841.6 1954.01   851.4 1953.67   890.8 1963.81   959.8  1962.5
  1038.7 1972.08  1058.4 1971.62  1107.7 1976.04  1166.8 1974.07  1196.4 1975.12
#Mann= 3 , 0 , 0
       0      .1       0   659.7    .045       0   674.7      .1       0
Bank Sta=659.7,674.7
XS Rating Curve= 0 ,0
Exp/Cntr=0.3,0.1

Type RM Length L Ch R = 1 ,36320.3 ,290.9,289.2,290.4
XS GIS Cut Line= 3
     1902284.123      232472.737     1902086.855      232995.929
     1901641.718      233430.204
#Sta/Elev= 30
       0 2113.42      20 2106.72    59.9 2078.98    99.8 2060.12   109.8 2059.04
   189.7 2025.39   209.7 2021.02   269.6 1996.15   399.4 1965.31   469.3 1953.08
   509.2 1936.29   519.2 1934.95   549.2 1907.37   559.2 1901.47   645.2 1887.15
     648 1886.89   660.2 1889.48   707.2 1905.38   746.7  1928.1   766.4 1935.44
   776.3 1943.54     875 2002.26   894.8 2006.29  1013.2 2061.01  1042.8 2067.03
  1082.3 2084.93  1141.6 2106.82  1151.4 2109.75  1161.3 2108.78    1181 2115.34
#Mann= 3 , 0 , 0
       0      .1       0   645.2    .045       0   660.2      .1       0
Bank Sta=645.2,660.2
XS Rating Curve= 0 ,0
Exp/Cntr=0.3,0.1

Type RM Length L Ch R = 1 ,36031.1 ,305.6,300,291.5
XS GIS Cut Line= 3
     1902223.645      232417.152     1901847.197      232830.492
     1901430.401       233193.26
#Sta/Elev= 30
       0 2155.74    59.9 2120.57    69.9 2115.46    79.9 2115.39   119.8 2092.26
   169.7 2067.01   199.7 2049.06   219.6 2041.97   279.5 2011.06   309.5 1999.55
   339.4 1992.44   399.3 1966.25   419.3 1955.61   439.3  1940.4   469.2 1927.18
   539.1  1887.3   549.1 1884.98   551.6 1885.09   566.6 1886.67   647.9 1902.52
   756.4 1927.45   874.8 1983.26   894.6 1990.46     934 2011.96   963.6 2025.36
   983.4 2039.08    1013 2051.22  1072.2 2084.05    1082 2094.49  1111.6 2112.73
#Mann= 3 , 0 , 0
       0      .1       0   551.6    .045       0   566.6      .1       0
Bank Sta=551.6,566.6
XS Rating Curve= 0 ,0
Exp/Cntr=0.3,0.1

Type RM Length L Ch R = 1 ,35731.1 ,305.8,300,293.4
XS GIS Cut Line= 3
     1901864.476      232174.241     1901611.929      232658.324
     1901359.083      233142.251
#Sta/Elev= 30
       0 2180.42    19.8 2173.02    49.6 2156.83   119.1 2107.55     139 2098.24
   168.8  2090.4   188.6 2080.88   208.5 2067.64   218.4 2058.05   248.2 2040.87
   297.8 1999.07   317.7 1987.55   337.5 1981.37   377.2 1960.38   426.9 1924.16
   446.7 1916.37   486.4 1893.28   536.1 1880.33   538.5 1880.35   553.5 1881.66
   655.2 1911.61   744.6 1948.13   764.4 1952.14   863.7 1992.08     963 2059.31
   972.9 2060.89   982.8 2066.88  1062.2 2128.07  1082.1 2137.06    1092 2144.34
#Mann= 3 , 0 , 0
       0      .1       0   538.5    .045       0   553.5      .1       0
Bank Sta=538.5,553.5
XS Rating Curve= 0 ,0
Exp/Cntr=0.3,0.1

Type RM Length L Ch R = 1 ,35431.1 ,291.6,300,312.8
XS GIS Cut Line= 3
     1901457.731      232012.002     1901335.765      232547.775
     1901232.309      233085.933
#Sta/Elev= 30
       0 2172.41      30 2151.12    59.9 2125.59    69.9 2119.56    79.9 2117.25
   119.9 2085.38   159.8 2058.33   169.8 2058.06   259.8 1999.68   269.7 1998.35
   349.7 1954.24   369.6 1948.31   429.6 1917.86   449.6 1909.85   469.6  1905.3
   489.5 1893.46   539.5 1876.22     542 1876.36     557 1876.81     669 1903.52
   738.8 1935.46   758.7 1940.53   828.5 1976.52   848.4 1983.19   928.1 2036.98
   938.1 2043.01     948 2044.17  1027.8 2102.83  1037.7 2103.74  1097.5 2145.48
#Mann= 3 , 0 , 0
       0      .1       0     542    .045       0     557      .1       0
Bank Sta=542,557
XS Rating Curve= 0 ,0
Exp/Cntr=0.3,0.1

Type RM Length L Ch R = 1 ,35131.1 ,291.4,300,301.3
XS GIS Cut Line= 3
     1901377.649      231977.239     1901066.636      232434.644
     1900692.204      232830.324
#Sta/Elev= 30
       0 2167.37     9.9  2164.5    29.6 2151.38    59.3 2119.95      79 2104.47
   118.5 2080.96     158 2063.27   227.2 2012.91   246.9 2005.19   266.7 1991.71
   316.1 1957.02   335.8 1940.57   395.1 1912.73   454.4 1891.21   543.2 1869.61
   545.6 1869.85   560.6 1872.63   592.7 1878.13   652.2 1896.52   691.8 1918.43
   711.6 1924.79   731.4 1938.94   850.3 2003.49   939.4 2060.99   959.2 2079.23
     979 2089.44  1048.4 2143.78  1058.3  2155.4  1078.1 2172.64  1097.9 2181.46
#Mann= 3 , 0 , 0
       0      .1       0   545.6    .045       0   560.6      .1       0
Bank Sta=545.6,560.6
XS Rating Curve= 0 ,0
Exp/Cntr=0.3,0.1

Type RM Length L Ch R = 1 ,34831.1 ,297.2,299.7,299.3
XS GIS Cut Line= 3
     1901313.605      231915.949      1900846.46      232233.026
     1900452.203      232605.994
#Sta/Elev= 30
       0 2146.78    39.6 2119.49    69.3 2093.03     109 2067.27   128.8 2061.74
   158.5 2042.16   227.8 2008.72   267.4  1984.8   287.2  1978.8     317 1963.56
   336.8 1957.33   356.6 1944.48   445.7 1898.72   465.5  1882.9   557.1 1865.14
   564.6 1864.96   572.1 1866.68   643.5 1897.73   673.1 1914.07   742.2 1941.96
   761.9 1952.94     831 1983.15   850.8 1994.38   860.6  2002.9   959.3 2059.63
   988.9  2083.9  1008.6 2093.09  1067.8 2131.46  1087.6 2149.95  1107.3 2163.26
#Mann= 3 , 0 , 0
       0      .1       0   557.1    .045       0   572.1      .1       0
Bank Sta=557.1,572.1
XS Rating Curve= 0 ,0
Exp/Cntr=0.3,0.1

Type RM Length L Ch R = 1 ,34531.1 ,310,290.3,284.1
XS GIS Cut Line= 3
     1901211.458      231751.761     1900705.965      231985.236
      1900273.82      232351.552
#Sta/Elev= 30
       0 2202.18    19.9  2187.7    39.8 2167.61   109.4 2121.18   129.3 2100.22
   149.1 2085.65     179 2064.75   188.9  2062.6   208.8 2050.04   228.7 2028.37
   278.4  1991.7   318.2 1970.81   377.8 1950.96   407.7 1938.09   457.4 1908.48
   477.3 1892.52   507.1 1877.54   549.3 1866.61   564.3 1863.86   566.7 1863.48
   636.3 1871.87     696 1884.27   805.3 1934.67   825.2 1938.98   864.9 1956.09
   954.4 2003.98   974.2  2010.7  1073.6 2065.42  1093.5 2079.63  1123.3 2091.28
#Mann= 3 , 0 , 0
       0      .1       0   549.3    .045       0   564.3      .1       0
Bank Sta=549.3,564.3
XS Rating Curve= 0 ,0
Exp/Cntr=0.3,0.1

Type RM Length L Ch R = 1 ,34240.7 ,296.3,300,296
XS GIS Cut Line= 3
     1900627.569      231267.666     1900504.904      231792.591
     1900211.132      232298.814
#Sta/Elev= 30
       0 2193.55      20 2184.44      30 2184.64   119.8 2129.19   129.8 2127.68
   139.8 2122.75   209.6 2072.25   229.6 2063.97   309.5 2004.72   319.4  1998.8
   329.4 1997.37   369.4 1968.79   379.3 1968.34   419.3 1935.67   429.3 1934.19
   509.1 1865.11   519.1 1860.78   529.1 1859.95   531.6 1860.08   546.6 1861.35
   618.4 1870.09   717.6 1877.63   747.4 1882.95   836.7 1929.73   866.4  1940.1
   945.8 1988.33   965.6 1995.27  1054.9 2053.76  1064.8 2054.96  1124.4 2101.15
#Mann= 3 , 0 , 0
       0      .1       0   531.6    .045       0   546.6     .06       0
Bank Sta=531.6,546.6
XS Rating Curve= 0 ,0
Exp/Cntr=0.3,0.1

Type RM Length L Ch R = 1 ,33940.7 ,296.6,297.5,299.3
XS GIS Cut Line= 3
     1900424.278      231221.537     1900212.389      231729.854
     1900022.398      232240.733
#Sta/Elev= 30
       0 2161.99    68.8 2119.36    88.5 2112.33   147.5 2074.85   167.2 2059.79
   186.8 2051.57   275.4 1998.39   285.2 1996.62     295 1991.15   373.7 1935.98
   383.5 1934.92   432.7  1898.8   452.4 1890.56   481.9 1866.53   491.7 1865.28
   511.4 1856.19   540.9 1855.28   543.2  1855.4   558.2 1856.81   639.9 1865.03
   699.4 1879.55   788.6 1928.07   808.4 1933.88   887.7 1982.64   907.5 1989.03
   947.1 2015.88   986.8 2046.63   996.7 2048.73    1066 2095.83  1095.8 2111.62
#Mann= 3 , 0 , 0
       0      .1       0   543.2    .045       0   558.2     .06       0
Bank Sta=543.2,558.2
XS Rating Curve= 0 ,0
Exp/Cntr=0.3,0.1

Type RM Length L Ch R = 1 ,33643.2 ,386.5,402,413.1
XS GIS Cut Line= 3
      1900314.56      231151.687     1899995.678      231502.954
     1899727.338      232083.105
#Sta/Elev= 30
       0 2140.58    49.4 2108.01   158.1 2043.13   177.9  2027.9   197.7 2019.83
   276.7 1971.39   296.5 1955.35   395.4 1909.47     425 1890.34   444.8 1882.98
   484.4  1856.4   494.4 1853.18   544.6 1852.33   559.6 1852.01   564.3 1851.98
   694.2 1866.74   714.1 1873.56   754.1 1895.61   764.1 1896.66     794  1907.7
   863.9 1958.87   873.9 1960.91   883.9 1967.35   923.9 2000.72   963.8 2028.28
   973.8 2030.24  1063.7 2085.25  1073.7 2087.63  1093.6 2101.86  1113.6 2106.42
#Mann= 3 , 0 , 0
       0      .1       0   544.6    .045       0   559.6      .1       0
Bank Sta=544.6,559.6
XS Rating Curve= 0 ,0
Exp/Cntr=0.3,0.1

Type RM Length L Ch R = 1 ,33240.6 ,233.7,225.6,222
XS GIS Cut Line= 3
     1900009.159      231241.767     1899608.111      231420.385
     1899495.211      231722.013
#Sta/Elev= 30
       0 1977.31    39.9 1954.42    59.9 1940.76    89.8 1927.37   109.8 1919.54
   129.7 1907.52   149.7 1891.81   229.5 1846.49   239.5 1844.96   253.3 1844.69
   268.3 1844.39   309.3 1843.45   319.3 1843.83   329.3 1845.32   369.2 1853.65
   448.8 1861.33   478.1 1867.29   487.8 1867.73   517.1  1876.1   556.1 1891.33
   575.7 1897.49   585.4 1899.34   595.2 1898.71   634.2 1907.23   653.7 1912.44
   663.5    1914   673.2 1914.53   692.8 1919.34   702.5 1918.89   761.1 1930.52
#Mann= 3 , 0 , 0
       0      .1       0   253.3    .045       0   268.3      .1       0
Bank Sta=253.3,268.3
XS Rating Curve= 0 ,0
Exp/Cntr=0.3,0.1

Type RM Length L Ch R = 1 ,33015.2 ,242.2,242.8,243.3
XS GIS Cut Line= 2
     1899964.671      230832.896     1899211.311      231656.966
#Sta/Elev= 30
       0 2148.51      10 2143.52    29.9 2128.69    79.8 2099.52    99.7  2092.5
   129.6 2075.28   149.5 2061.68   209.4 2036.75   219.3 2034.71   229.3 2028.82
   249.2 2015.33   269.2  1998.4     339 1949.07   358.9 1941.27   468.5 1855.08
   488.5 1846.34   528.4 1843.55     530 1843.55     545 1844.03   717.8 1864.12
   757.6 1870.35   767.6 1873.13   797.5 1887.22   827.4 1897.13   837.4 1902.22
   867.3 1909.52   877.3 1910.91   947.1 1911.34  1046.8 1918.27  1116.5 1935.54
#Mann= 3 , 0 , 0
       0      .1       0     530    .045       0     545      .1       0
Bank Sta=530,545
XS Rating Curve= 0 ,0
Exp/Cntr=0.3,0.1

Type RM Length L Ch R = 1 ,32772   ,303.8,306.7,309.7
XS GIS Cut Line= 3
     1899832.027      230665.649      1899447.45      231055.456
     1899057.562      231453.159
#Sta/Elev= 30
       0 2129.08   159.3 2057.42   179.2 2045.25   199.1 2039.44   268.8 2008.79
   278.8 2003.03   308.6 1979.44   328.6 1970.66   368.4 1944.63   388.3 1930.88
   408.2 1913.63     448 1890.74   477.9 1877.32   507.8 1859.53   517.7 1849.98
   527.7 1844.46   537.6 1843.38   537.8 1843.42   552.8 1846.57   577.4 1851.94
   716.7 1860.86   806.2 1886.84     836 1898.27   855.9 1910.84   945.4 1955.21
   965.3 1970.47   985.2 1978.01  1064.7  2022.5  1084.6 2037.54  1104.5 2045.86
#Mann= 3 , 0 , 0
       0      .1       0   537.8    .045       0   552.8      .1       0
Bank Sta=537.8,552.8
XS Rating Curve= 0 ,0
Exp/Cntr=0.3,0.1

Type RM Length L Ch R = 1 ,32465.3 ,345.9,366,386
XS GIS Cut Line= 3
     1899707.531      230684.008     1899321.649      230780.057
     1898798.063      231193.996
#Sta/Elev= 30
       0 2077.64     9.9 2069.28    19.9 2064.21    69.6 2042.76    89.5 2030.52
   159.1 1999.27     169 1991.67   238.6 1949.91   248.5  1938.2   318.1 1898.02
     338 1881.69   397.7 1849.04   417.6 1844.53   506.5 1838.87   507.2  1838.8
   521.5 1840.44   537.1 1844.32   586.9  1845.8   636.7 1858.61   666.6 1869.72
   756.3 1910.43   806.1  1928.2   816.1 1933.44     826 1941.54   905.7  1977.3
   935.6 1998.85  1005.3 2040.72  1015.3 2044.13  1035.2 2059.91  1065.1 2079.97
#Mann= 3 , 0 , 0
       0     .06       0   506.5    .045       0   521.5     .06       0
Bank Sta=506.5,521.5
XS Rating Curve= 0 ,0
Exp/Cntr=0.3,0.1

Type RM Length L Ch R = 1 ,32099.4 ,257.8,258.7,260.5
XS GIS Cut Line= 3
     1899635.073       230621.66       1899338.5      230581.218
     1898616.707      230433.965
#Sta/Elev= 30
       0 2038.51      10 2032.38      20 2022.58    89.8 1987.54    99.8 1976.03
   169.6 1932.69   179.6 1922.77   219.5 1901.38   249.4  1882.2   259.4 1869.86
   269.4 1861.76   299.3 1841.93   319.2 1838.14   478.5 1829.94   491.3 1830.66
   506.3 1837.02     578 1857.79   657.7 1893.09   667.6 1900.62   727.4 1928.63
   737.3 1934.22   757.2 1950.69     817 1981.81   836.9 1997.23   896.6 2030.65
   916.5 2047.42   926.5 2052.84   936.4 2054.65  1006.1  2097.7    1036 2111.43
#Mann= 3 , 0 , 0
       0     .06       0   491.3    .045       0   506.3     .06       0
Bank Sta=491.3,506.3
XS Rating Curve= 0 ,0
Exp/Cntr=0.3,0.1

Type RM Length L Ch R = 1 ,31840.7 ,116.1,115.9,114.7
XS GIS Cut Line= 3
     1899747.122      230421.824     1899215.803      230293.123
     1898691.648      230140.659
#Sta/Elev= 30
       0  2015.4    29.8 2014.16    49.7 2010.81   109.3 1981.29   119.3 1975.98
   139.2 1960.47   198.8 1928.68   218.7 1913.61   288.2 1876.19   298.2  1864.4
     338  1837.2   357.8 1833.85     497  1832.5   539.2 1827.12   546.7 1826.28
   554.2 1828.54   626.1 1852.44   645.9 1861.23   705.5 1880.36   725.3  1889.5
   794.8 1910.43   804.7 1916.11   824.6 1923.16   874.2 1945.49   894.1 1958.27
   963.5 1991.02   973.5 1999.19    1033 2029.45  1052.9  2043.1  1092.6 2062.02
#Mann= 3 , 0 , 0
       0     .06       0   539.2    .045       0   554.2     .06       0
Bank Sta=539.2,554.2
XS Rating Curve= 0 ,0
Exp/Cntr=0.3,0.1

Type RM Length L Ch R = 1 ,31724.8 ,185.6,184,182.3
XS GIS Cut Line= 2
     1899655.293       230276.22     1898659.415      230045.365
#Sta/Elev= 30
       0 1930.97    29.8 1915.21    39.7 1906.52    49.6 1901.74   119.1  1872.6
     139 1861.06   178.6 1844.06   198.5 1837.45   208.4 1835.84     410 1824.34
   416.8 1824.17     425 1824.74   446.6 1830.52   486.3 1850.11     526 1867.68
     536 1873.16   545.9 1880.47   615.4 1914.63   625.3 1923.15     665 1943.16
   694.8 1955.05   774.2  1991.9     794 2004.35   853.6 2030.09   863.5 2035.11
   873.4 2042.62   942.9 2075.68   952.8 2083.13   972.7 2089.08  1022.3 2115.15
#Mann= 3 , 0 , 0
       0     .06       0     410    .045       0     425     .06       0
Bank Sta=410,425
XS Rating Curve= 0 ,0
Exp/Cntr=0.3,0.1

Type RM Length L Ch R = 1 ,31540.7 ,223,224.6,226.4
XS GIS Cut Line= 3
     1899825.531      230087.873     1899286.345      230002.234
      1898746.66      229919.033
#Sta/Elev= 30
       0 1866.64    79.4 1859.13     129 1856.95   168.8  1853.2   337.5 1842.26
   347.4  1841.1   377.2 1829.64   387.1 1828.02   456.6  1826.6   538.4 1820.36
     546 1819.66   553.4 1820.86   615.4  1843.3   625.4 1849.87   665.1 1869.21
   694.9 1888.44   704.8 1900.78   714.7  1910.3   724.7 1916.95   774.3 1944.72
   794.2 1961.92   853.7 1991.45   873.6 2005.42   933.2    2029   943.1 2033.42
     953 2039.77   982.8 2049.45  1022.5 2064.58  1042.4 2076.69    1092 2096.09
#Mann= 3 , 0 , 0
       0     .06       0   538.4    .045       0   553.4     .06       0
Bank Sta=538.4,553.4
XS Rating Curve= 0 ,0
Exp/Cntr=0.3,0.1

Type RM Length L Ch R = 1 ,31316   ,290.4,290.3,290.2
XS GIS Cut Line= 2
     1899831.242       229899.68      1898768.12      229650.207
#Sta/Elev= 30
       0 1928.71    49.6 1907.76    69.5 1895.93     139 1871.47   148.9 1864.73
   168.8  1859.2   258.1 1841.94   297.8 1838.68   387.2 1835.25   486.4 1824.03
   511.5 1819.03   516.2 1818.61   526.5    1820   555.9 1832.01   575.8 1843.56
   605.6 1854.14   625.4  1864.3   635.4 1870.71   645.3 1881.11   655.2 1895.01
   724.7 1943.38   734.6 1956.18     814 2003.96   843.8 2015.69   893.4 2028.72
     963 2050.53   972.9 2054.88  1032.4 2092.67  1062.2  2105.7    1092 2112.99
#Mann= 3 , 0 , 0
       0     .06       0   511.5    .045       0   526.5     .06       0
Bank Sta=511.5,526.5
XS Rating Curve= 0 ,0
Exp/Cntr=0.3,0.1

Type RM Length L Ch R = 1 ,31025.7 ,311.7,310.1,308.5
XS GIS Cut Line= 2
     1899925.771      229621.303     1898861.029      229376.342
#Sta/Elev= 30
       0 2024.26     9.9 2013.66    79.5 1974.74    89.4 1964.59    99.3 1957.85
   158.9 1922.76   178.8 1905.44   238.4  1872.6   248.3 1865.36   258.2 1854.65
     288 1836.72   357.6 1824.36   506.6 1822.36   537.7 1818.62   546.3 1818.56
   552.7 1819.53   576.1 1826.04   655.5 1866.42   665.5 1875.82     735 1913.27
   754.9 1928.78   824.4  1966.9   844.2  1983.6   913.8 2022.97   923.7 2033.76
   993.2 2072.49  1003.2 2082.02  1013.1 2088.46  1072.7 2118.81  1092.6  2131.4
#Mann= 3 , 0 , 0
       0     .06       0   537.7    .045       0   552.7     .06       0
Bank Sta=537.7,552.7
XS Rating Curve= 0 ,0
Exp/Cntr=0.3,0.1

Type RM Length L Ch R = 1 ,30715.6 ,387.8,374.9,359.1
XS GIS Cut Line= 2
     1900068.136      229298.877     1899137.976      229152.276
#Sta/Elev= 30
       0 1951.68    69.4 1927.55    79.3 1922.11    99.1 1914.09   168.5 1892.37
     228 1881.63   247.8 1875.94   307.3 1865.21   317.2 1862.78   327.1 1858.44
   396.5 1842.34   406.4 1837.73     456 1824.58   465.9 1823.24   545.2 1821.79
   555.1  1820.8   561.8 1818.74   574.9 1816.16   576.8 1816.17   594.7 1816.64
   693.8  1823.2   703.8  1824.5   713.7  1827.4   723.6 1833.36   733.5 1841.92
   802.9 1875.64   812.8 1884.54   882.2 1926.17   892.1 1938.02   941.6 1968.48
#Mann= 3 , 0 , 0
       0     .06       0   561.8    .045       0   576.8     .06       0
Bank Sta=561.8,576.8
XS Rating Curve= 0 ,0
Exp/Cntr=0.3,0.1

Type RM Length L Ch R = 1 ,30340.7 ,306.2,300,293
XS GIS Cut Line= 3
     1899948.567      228639.323     1899478.713      228846.963
     1898853.266      229221.642
#Sta/Elev= 30
       0 2045.29    39.5 2029.89    59.3 2017.87   128.4 1986.69   158.1 1969.21
   187.7 1961.17   237.1 1941.82   306.2 1923.58     326 1911.59   395.2 1882.73
   414.9 1866.62   444.5 1847.66   493.9 1820.49   506.2 1816.18   521.2 1814.12
   523.7    1814   663.5 1822.12   743.4 1831.28   773.4 1856.95   823.3 1882.69
   843.3  1888.2   933.2 1943.13   953.1 1961.63  1013.1 2004.88    1033 2015.83
    1043 2025.84  1122.9 2071.64  1132.9 2080.52  1232.8  2119.5  1242.8  2120.6
#Mann= 3 , 0 , 0
       0     .06       0   506.2    .045       0   521.2     .06       0
Bank Sta=506.2,521.2
XS Rating Curve= 0 ,0
Exp/Cntr=0.3,0.1

Type RM Length L Ch R = 1 ,30040.7 ,96.5,88.4,83.8
XS GIS Cut Line= 3
     1899674.114      228301.518     1899274.434      228628.554
     1898800.038      229161.606
#Sta/Elev= 30
       0 2056.51    19.9 2057.31    49.7  2051.8    79.4 2038.71   119.2 2014.78
     139 2000.08   208.6 1963.73   228.4 1957.23   248.3 1941.48   317.8 1901.32
   337.7 1887.08   397.2 1865.36   466.8  1831.9   508.9 1815.51   523.9  1812.1
   526.3  1811.8   724.6 1822.87   744.4 1828.52   764.2 1840.21   774.1 1843.25
   813.8 1869.29   873.2 1911.56   883.1 1921.11     903 1931.52  1021.9 2020.52
  1031.8 2022.42  1140.8 2085.71  1160.6 2088.89  1190.4  2103.5    1230 2106.62
#Mann= 3 , 0 , 0
       0     .06       0   508.9    .045       0   523.9     .06       0
Bank Sta=508.9,523.9
XS Rating Curve= 0 ,0
Exp/Cntr=0.3,0.1

Type RM Length L Ch R = 1 ,29952.3 ,501.2,495.1,489.1
XS GIS Cut Line= 4
     1899758.083      227979.465     1899282.892       228439.49
     1899104.274      228747.858     1898734.424      229137.624
#Sta/Elev= 30
       0 1954.51    19.7 1958.51    59.2 1954.99   108.6 1956.25   157.9 1951.14
   217.2 1938.58   335.6 1966.36   365.2 1970.23   394.9 1962.72   473.8 1956.24
   533.1 1924.13   602.2 1880.09     701 1849.56   740.6  1831.8   822.6 1812.07
   829.7 1811.69   837.6 1812.01  1047.6 1823.78  1057.6  1827.5  1107.3 1861.32
  1127.2 1868.46  1226.7 1944.48  1246.6 1954.02  1306.3 1996.34    1366 2027.43
  1385.9 2030.99  1445.6 2071.88  1475.5 2078.44  1515.3 2071.52  1555.1 2071.37
#Mann= 3 , 0 , 0
       0     .06       0   822.6    .045       0   837.6     .06       0
Bank Sta=822.6,837.6
XS Rating Curve= 0 ,0
Exp/Cntr=0.3,0.1

Type RM Length L Ch R = 1 ,29457.2 ,318,316.4,313.8
XS GIS Cut Line= 4
     1899087.424      227908.692     1898798.373      228294.785
     1898703.227      228646.754     1898482.088      229052.459
#Sta/Elev= 30
       0 1882.56    59.1 1887.96   167.3 1869.83     187 1870.87   255.9 1859.32
   295.3 1859.77   393.7 1851.86   433.1 1853.73   482.3 1845.15   511.9 1835.92
   521.7 1836.08   580.8 1816.71   689.2 1815.27   754.2  1810.7   768.1 1809.77
   769.2 1809.95   797.6 1817.85     837 1822.14   905.9 1857.61   915.7 1861.07
   935.4 1861.83  1023.9  1905.7  1033.7 1905.71  1063.2 1916.46  1092.7 1921.17
  1122.2 1940.23  1141.8 1947.92  1240.2 2019.73  1259.8 2027.45    1309 2056.39
#Mann= 3 , 0 , 0
       0     .06       0   754.2    .045       0   769.2     .06       0
Bank Sta=754.2,769.2
XS Rating Curve= 0 ,0
Exp/Cntr=0.3,0.1

Type RM Length L Ch R = 1 ,29140.7 ,291.4,300.1,308.2
XS GIS Cut Line= 3
     1898526.227      227942.878     1898423.176        228480.1
     1898343.987      229020.145
#Sta/Elev= 30
       0 2064.11    69.6 2035.64    99.5 2028.28   119.4 2019.91   139.2 2007.17
     179 1974.92   198.9 1968.18   268.5 1912.22   288.4 1906.01     358  1868.1
   377.9 1860.12   387.9 1860.07   407.8 1849.91   477.4 1839.57   539.5 1811.43
     547 1809.66   554.5 1809.66   596.6 1817.22   695.9  1827.4   705.8 1830.97
   765.3 1866.82   785.2 1867.96   874.5 1929.18   884.4 1929.35   963.8 1987.64
   973.8 1989.17   983.7 1995.34  1053.1 2043.95  1063.1 2050.22  1092.8 2061.13
#Mann= 3 , 0 , 0
       0      .1       0   539.5    .045       0   554.5      .1       0
Bank Sta=539.5,554.5
XS Rating Curve= 0 ,0
Exp/Cntr=0.3,0.1

Type RM Length L Ch R = 1 ,28840.7 ,321.4,310.6,301.3
XS GIS Cut Line= 3
     1898443.245      227910.531     1898144.916      228374.439
     1897879.396      228850.408
#Sta/Elev= 30
       0 2079.09    19.7 2066.94    39.4 2061.32    88.6 2038.22   137.9 2005.89
   157.6 1996.67   177.3  1992.5     197 1983.31   216.7 1971.25   246.2  1948.9
   256.1 1942.84   265.9 1940.95   315.2 1903.38   354.6 1879.53   374.3  1874.1
   413.7    1855   462.9 1840.41   502.3 1832.27     522 1823.51   544.1 1809.86
   551.6 1807.84   559.1  1808.3   591.2 1816.17   640.7 1816.93   690.3 1839.65
   799.3 1851.82   858.8 1854.38   908.3 1866.59  1037.1 1880.18  1096.6 1893.04
#Mann= 3 , 0 , 0
       0      .1       0   544.1    .045       0   559.1      .1       0
Bank Sta=544.1,559.1
XS Rating Curve= 0 ,0
Exp/Cntr=0.3,0.1

Type RM Length L Ch R = 1 ,28530.1 ,349.8,345.9,341.9
XS GIS Cut Line= 3
      1897964.49      227682.103      1897850.58      228520.373
     1897743.447       228774.63
#Sta/Elev= 30
       0 2141.04    49.8 2126.76    69.7 2124.66    79.6 2118.53   139.3 2064.36
   159.2 2054.63   238.9 1995.36   258.8 1987.35   298.6 1954.15   308.5  1949.3
   348.3 1942.82   358.3 1937.42   378.2 1922.07     428 1871.75   437.9 1864.99
   467.8 1857.13   507.6  1829.6   527.5 1812.07     533 1811.73     548  1806.5
   557.4 1806.42   617.1 1816.47   666.8 1815.35   716.6 1830.34   806.2 1847.51
   885.4 1851.18   924.8 1857.96  1023.3  1897.7  1062.8 1906.69  1121.9 1929.17
#Mann= 3 , 0 , 0
       0      .1       0     533    .045       0     548      .1       0
Bank Sta=533,548
XS Rating Curve= 0 ,0
Exp/Cntr=0.3,0.1

Type RM Length L Ch R = 1 ,28184.2 ,235.4,243.4,250.5
XS GIS Cut Line= 2
      1897526.14      227669.619     1897576.963      228770.467
#Sta/Elev= 30
       0 1945.81    69.5 1939.22   158.8 1926.52   188.6 1917.26   258.1 1903.08
   327.6 1876.82   377.3 1862.68   426.9 1838.66   446.8 1833.65   476.6 1819.05
   486.5 1815.97   536.1 1810.04   549.4 1804.01     556 1802.89   564.4 1804.21
   585.8 1810.16     695 1812.54   704.9 1815.86   724.8 1827.71   734.7 1827.82
   774.4 1853.09   794.2  1856.7   814.1 1868.22     824    1869   853.8 1889.46
   913.4 1918.23   933.2 1922.19   992.8 1947.75  1052.4 1960.66    1102 1979.48
#Mann= 3 , 0 , 0
       0     .06       0   549.4    .045       0   564.4     .06       0
Bank Sta=549.4,564.4
XS Rating Curve= 0 ,0
Exp/Cntr=0.3,0.1

Type RM Length L Ch R = 1 ,27940.7 ,291.5,299.9,308.3
XS GIS Cut Line= 3
     1897481.988       227660.12     1897311.282      228198.175
     1897165.245      228720.897
#Sta/Elev= 30
       0 1938.67    49.5 1923.54   178.3 1895.32   247.6 1874.11     307 1867.45
   356.5 1844.19   376.3 1838.44   415.9 1819.01   524.9 1812.74     557 1800.27
   564.5 1800.07     572  1800.7   594.1 1807.15   623.7 1811.54   653.3 1833.79
   663.2 1834.47   692.8 1857.96   712.5 1863.62     752 1895.55   771.7 1903.28
   850.7 1964.53   860.5 1965.45     900 1993.45   949.3 2024.12   969.1    2030
   978.9  2035.7    1048 2082.58  1057.9 2083.94  1087.5 2103.97  1107.2 2110.91
#Mann= 3 , 0 , 0
       0      .1       0     557    .045       0     572      .1       0
Bank Sta=557,572
XS Rating Curve= 0 ,0
Exp/Cntr=0.3,0.1

Type RM Length L Ch R = 1 ,27640.7 ,245.9,246.3,247.5
XS GIS Cut Line= 3
     1897403.958      227618.837      1897046.22      228060.383
     1896721.392      228494.347
#Sta/Elev= 30
       0 1953.41    29.9 1951.69   119.6 1921.32   139.6 1918.01   239.3 1875.48
   279.2 1867.26   358.9 1831.78   378.8 1826.56   398.8 1815.46   528.4 1806.52
   558.3 1797.42   560.8 1797.52   575.8 1800.05   617.6 1810.34   627.4 1816.94
     657 1848.63   666.8 1855.88   686.6 1861.58   716.1 1889.86   735.8 1897.77
   755.5 1911.73   804.8 1955.86   854.1 1979.99   923.1 2021.62   952.6 2036.76
   972.4 2041.73  1001.9 2056.21  1011.8 2058.57  1041.4 2056.12  1110.4 2043.71
#Mann= 3 , 0 , 0
       0      .1       0   560.8    .045       0   575.8      .1       0
Bank Sta=560.8,575.8
XS Rating Curve= 0 ,0
Exp/Cntr=0.3,0.1
